--- Vall Creek.prj (project) ---

Proj Title=Vall Creek
Current Plan=p01
Default Exp/Contr=0,0
English Units
Geom File=g01
Flow File=f01
Plan File=p01
BEGIN DESCRIPTION:
END DESCRIPTION:
DSS Export Rating Curves= 0
DSS Export Rating Curve Sorted= 0
DSS Export Volume Flow Curves= 0
DXF OffsetX= 0
DXF OffsetY= 0
DXF ScaleX= 0
DXF ScaleY= 0

--- Vall Creek.p01 (plan) ---

Plan Title=Floodplain
Program Version=4.00
Geom File=g01
Flow File=f01
K Sum by GR=0
Std Step Tol=0.01
Critical Tol=0.01
Num of Std Step Trials=20
Max Error Tol=0.3
Flow Tol Ratio=0.001
Split Flow NTrial=30
Split Flow Tol=0.02
Split Flow Ratio=0.02
Log Output Level=0
Friction Slope Method=1
Unsteady Friction Slope Method=2
Unsteady Bridges Friction Slope Method=1
Global Log Level=0
CheckData=False
Run HTab=0
Run UNet=0
Run PostProcess=0
UNET Theta=0
UNET Theta Warmup=0
UNET ZTol=0
UNET ZSATol=0
UNET MxIter=0
UNET MaxInSteps=0
UNET DtIC=0
UNET DtMin=0
UNET MaxCRTS=0
UNET WFStab=0
UNET SFStab=0
UNET WFX=0
UNET SFX=0
UNET DSS MLevel=0
UNET DZMax Abort=0
UNET Convert EG Bridges=0
UNET Use Existing IB Tables=0
UNET Froude Limit=0
UNET Froude Power=0
Write IC File=0
Echo Input=False
Echo Output=False
Write Detailed=0

--- Vall Creek.f01 (steady flow) ---

Flow Title=NFF Regression Equation
Program Version=4.00
Number of Profiles=1
Profile Names=P100yr
River Rch & RM=Vall Creek,Main      ,17631.4
596.8272
River Rch & RM=Vall Creek,Main      ,16240
652.4867
River Rch & RM=Vall Creek,Main      ,14668.2
700.6036
River Rch & RM=Vall Creek,Main      ,13255.8
777.6512
River Rch & RM=Vall Creek,Main      ,11162.3
861.2285
River Rch & RM=Vall Creek,Main      ,10427.8
1256.259
Boundary for River Rch & Prof#=Vall Creek,Main      ,1
Up Type=0
Dn Type=3
Dn Slope=0.017474

--- Vall Creek.g01 (geometry) ---

Geom Title=USGS 10m DEM
Program Version=4.00

River Reach=Vall Creek      ,Main
Reach XY= 30
     1766174.937       86302.471      1766652.46       86607.399
     1766919.546        86585.72     1767218.763       86745.302
     1767377.514       86656.368     1768002.125       86796.342
     1768621.759       86739.484     1768804.614       86860.002
     1769059.485       86752.906     1769703.927       86837.561
     1770219.268        86692.87     1770785.264       86287.334
     1771516.684       86132.738     1772115.118       85546.771
     1772693.604       85377.215     1774059.198       85958.195
     1774449.011       85755.392     1774525.417       85867.966
     1774814.721        85753.73     1775426.454       86015.545
     1775773.878       85900.014     1776282.547       86249.101
     1777013.967       86441.929     1777557.694       86347.951
     1778344.917       86513.204     1778929.866       86066.838
     1780055.175       85845.492     1780575.137       85270.791
      1781270.39       85130.592     1781552.451       85238.641

Type RM Length L Ch R = 1 ,17631.4 ,122.7,121.9,121.2
XS GIS Cut Line= 5
     1765895.445       86721.403     1766059.298       86453.199
     1766190.014       86302.413     1766351.155       86116.532
     1766488.053       85958.615
#Sta/Elev= 30
     9.8 2007.97   186.6 2007.52   206.3 2002.81   225.9 2007.47   245.5 1999.79
   265.2 1996.29   384.1 1985.77   491.4 1983.15   503.9 1982.78  509.85 1984.43
   572.9 2020.83   602.4  2028.4   622.1  2039.1   651.6 2047.57   671.3 2060.89
     691 2062.25   700.8 2073.92   710.7 2080.18   730.3 2082.57     750 2097.13
   779.8 2105.84   799.7 2121.49   819.6 2123.39   839.5 2138.28   859.4 2141.98
   889.2 2159.57   919.1  2169.4     929  2178.7   958.9 2187.42   968.9 2194.84
#Mann= 3 , 0 , 0
     9.8      .1       0   491.4    .045       0  509.85      .1       0
#XS Ineff= 2 , 0
          454.51 2004.11
Permanent Ineff=
       F       F
Bank Sta=491.4,509.85
XS Rating Curve= 0 ,0
Exp/Cntr=0.3,0.1

Type RM Length L Ch R = 1 ,17509.4 ,99,95.7,92.4
XS GIS Cut Line= 4
     1765978.209       86731.291     1766210.639       86468.057
     1766403.864       86230.026     1766541.082         86031.2
#Sta/Elev= 30
      10 2033.42    50.2 2029.46    70.2 2034.28    90.3  2025.7   110.4 2031.63
   140.5 2024.65   250.8 2026.97   270.9 2017.46     291 2018.03   321.1 2001.82
   341.1 2001.04   361.1 1988.38   437.6 1982.77   450.1 1980.91   462.6 1981.64
   479.7 1988.66   489.6 2000.63   558.9 2025.95   578.6 2039.48   608.3 2046.42
   618.2 2056.15   687.9 2082.82   708.1 2099.04   728.2 2100.74   748.3 2115.63
   768.5 2119.16   798.7 2138.16   818.8  2140.9   838.9 2157.19   899.3 2181.04
#Mann= 3 , 0 , 0
       0      .1       0   437.6    .045       0   462.6      .1       0
Bank Sta=437.6,462.6
XS Rating Curve= 0 ,0
Exp/Cntr=0.3,0.1

Type RM Length L Ch R = 1 ,17413.8 ,217.4,215.5,213.7
XS GIS Cut Line= 4
     1766109.913       86783.297     1766303.353       86527.956
     1766415.548       86338.384     1766601.251       86048.224
#Sta/Elev= 30
      10 2088.26      20 2081.92      40 2086.94    70.1 2079.96    90.1 2082.97
   110.1 2073.54   130.1 2071.83   320.3 1994.34   360.4 1982.64   400.4 1978.47
   420.5 1977.63  424.69 1979.41   480.5 2006.12   500.6 2008.26   520.6 2021.02
   540.6 2023.99   560.3 2036.95     580 2039.37   599.7 2054.34   619.4  2055.9
   678.4 2090.17     708 2099.37   717.8 2112.27   737.5 2113.16   757.2 2127.89
   786.7 2137.27   806.4 2153.03   826.1 2154.91   835.9    2167   885.1 2190.96
#Mann= 3 , 0 , 0
      10      .1       0   400.4    .045       0  424.69      .1       0
Bank Sta=400.4,424.69
XS Rating Curve= 0 ,0
Exp/Cntr=0.3,0.1

Type RM Length L Ch R = 1 ,17198.2 ,50.4,49.7,49
XS GIS Cut Line= 4
     1766267.368       86929.242     1766473.261        86687.82
     1766672.912       86278.826     1766764.877       86114.706
#Sta/Elev= 30
     9.9 2148.42    69.4 2137.06    89.2 2122.09   109.1 2120.49   138.8 2104.23
   158.6 2101.35   178.5 2086.31   198.3 2085.82   347.6 2006.26   456.5 1977.92
     469 1974.76   481.5 1975.24   539.8 1998.92   590.4 2009.51   610.6 2025.42
   630.8  2030.4   651.1 2051.69   671.3 2053.94   691.5 2072.84   711.7  2079.6
     732 2095.53   742.1 2095.59   762.3 2116.28   782.3 2118.78   802.1 2135.65
   821.9 2143.58   841.7 2162.68   861.5 2165.31   881.3 2186.24   960.5 2210.06
#Mann= 3 , 0 , 0
       0      .1       0   456.5    .045       0   481.5      .1       0
Bank Sta=456.5,481.5
XS Rating Curve= 0 ,0
Exp/Cntr=0.3,0.1

Type RM Length L Ch R = 1 ,17148.5 ,11.7,11.5,11.3
XS GIS Cut Line= 4
     1766383.855       86900.159     1766555.682       86637.529
     1766622.736       86488.054     1766712.142       86225.424
#Sta/Elev= 30
     9.8 2133.31    29.4 2131.08    39.2 2120.56    68.7 2111.06    88.3 2093.55
   107.9 2090.14   127.5 2069.67   147.1 2065.25     206  2029.7   235.4 2019.44
   245.2 2008.98   274.6 2007.24   378.4 1976.96   390.9 1974.75  396.33 1977.64
   419.9 1982.41   439.1 1993.71   497.5 2002.08   527.2 2015.23     547 2035.39
   566.8  2037.8   576.8 2049.92   636.2  2081.8     656 2099.94   675.8 2100.79
   685.7 2115.99   705.6 2121.38   725.4 2139.54   745.2 2145.47   755.1 2154.34
#Mann= 3 , 0 , 0
     9.8      .1       0   378.4    .045       0  396.33      .1       0
Bank Sta=378.4,396.33
XS Rating Curve= 0 ,0
Exp/Cntr=0.3,0.1

Type RM Length L Ch R = 1 ,17137   ,49.4,47.6,45.9
XS GIS Cut Line= 4
     1766431.868        86949.72     1766569.652       86636.132
     1766636.706       86482.466      1766751.11       86176.819
#Sta/Elev= 30
    10.1 2144.79    40.3 2133.78    60.4 2113.38    80.6 2110.33    90.7 2098.76
   171.3 2055.01   191.4  2051.1   241.8  2025.1   261.9 2024.49   282.1 2011.68
   302.2 2011.23   399.1 1973.81   411.6 1973.42  417.97 1976.29   470.7 1994.56
   520.1 2000.02   559.6 2020.34   579.4 2038.02   599.2 2045.01   609.1 2059.85
   628.9 2061.56   688.2 2103.86     708  2108.8   717.9  2120.6   737.6 2123.63
   757.4  2143.9   777.2 2149.79   787.1 2161.97   806.9 2168.64   836.5 2192.16
#Mann= 3 , 0 , 0
    10.1      .1       0   399.1    .045       0  417.97      .1       0
Bank Sta=399.1,417.97
XS Rating Curve= 0 ,0
Exp/Cntr=0.3,0.1

Type RM Length L Ch R = 1 ,17089.4 ,64.8,57.4,49.9
XS GIS Cut Line= 4
     1766482.015        86916.06     1766611.832         86669.8
     1766676.817       86490.279     1766751.955       86237.036
#Sta/Elev= 30
     9.9 2116.16    19.9 2101.81    39.8  2098.1    59.7 2081.29    99.4    2065
   119.3 2069.06   139.2 2057.14   159.1 2058.26   198.8 2045.64   218.7  2033.7
   238.6 2035.49   248.6 2023.19   268.4 2020.02   308.5    2000   328.6 1981.64
  355.74 1975.56   358.8  1973.4   371.3 1974.14     399  1987.8   488.9 2001.46
   508.4 2021.26     528 2028.02   537.8 2041.12   557.4 2047.65   576.9 2065.09
   635.6 2091.95   645.4 2104.49     665 2106.26   684.5 2123.42   733.5 2149.27
#Mann= 3 , 0 , 0
     9.9      .1       0  355.74    .045       0   371.3      .1       0
Bank Sta=355.74,371.3
XS Rating Curve= 0 ,0
Exp/Cntr=0.3,0.1

Type RM Length L Ch R = 1 ,17032   ,91.4,89.5,87.6
XS GIS Cut Line= 4
     1766527.744       86980.606     1766689.502       86706.088
     1766695.102       86456.856     1766814.035       86148.813
#Sta/Elev= 30
      10 2129.51    59.7  2108.5    79.7 2113.94    99.6 2104.53   119.5 2109.04
   199.1 2092.57   219.1 2076.13     239 2071.78   278.8 2048.47   298.7 2031.18
   318.6 2031.04   328.6    2018   348.5 2013.72   405.8    1972   418.3 1970.87
  424.51  1973.9   468.2 1988.78     548 2001.78     608 2047.65     628 2049.23
     638 2065.12     698 2090.25     718 2107.76     738 2111.06     748 2123.79
   768.1 2126.69   788.1 2147.33   808.1 2153.73   858.1 2189.53   898.1 2200.78
#Mann= 3 , 0 , 0
      10      .1       0   405.8    .045       0  424.51      .1       0
Bank Sta=405.8,424.51
XS Rating Curve= 0 ,0
Exp/Cntr=0.3,0.1

Type RM Length L Ch R = 1 ,16942.5 ,66.8,67,67.3
XS GIS Cut Line= 4
     1766692.585       86989.565     1766784.785       86680.835
     1766772.212       86502.023      1766860.09       86218.177
#Sta/Elev= 30
    10.1 2167.91    80.6 2141.16   100.7 2123.55   161.1 2093.08   171.2 2079.32
   191.3 2077.84   201.4 2061.06   221.5 2055.59   241.7 2037.44   261.8 2032.19
   281.9 2015.95   389.4 1972.14   401.9 1970.85   414.4 1972.57   481.5 1994.08
   501.5  1994.5   511.4    2006   531.2 2009.89   570.8 2032.29   590.6 2049.98
   640.1 2070.23   659.9 2088.77   679.7 2091.85   689.6 2104.72   709.5  2107.2
   729.3 2124.49   749.1 2131.16   768.9 2150.14   788.7 2156.69   798.6 2172.14
#Mann= 3 , 0 , 0
    10.1      .1       0   389.4    .045       0   414.4      .1       0
#XS Ineff= 2 , 0
          388.42 1992.38
Permanent Ineff=
       F       F
Bank Sta=389.4,414.4
XS Rating Curve= 0 ,0
Exp/Cntr=0.3,0.1

Type RM Length L Ch R = 1 ,16875.5 ,156.6,176.9,197.2
XS GIS Cut Line= 4
     1766700.929       87023.163     1766850.518       86704.741
     1766836.337       86446.711     1766944.663       86195.239
#Sta/Elev= 30
    10.1 2175.11    50.3 2167.81   130.7 2133.77   140.7 2119.44   160.8  2116.5
   180.9 2096.39     201 2089.85   221.1 2071.43   241.2 2068.52   251.3 2052.72
   271.4  2047.9   331.7  2004.7   351.8 2004.68   371.7  1991.1   468.5 1968.82
     481 1968.13   484.5 1970.11     620 2031.78   639.6 2049.58   659.1 2049.94
   668.9  2061.9   737.4 2091.06   747.1 2104.82   766.7 2105.79   786.2 2121.53
   805.8 2125.23   825.4 2142.61   844.9 2142.38   864.5 2153.17     884 2146.06
#Mann= 3 , 0 , 0
    10.1      .1       0   468.5    .045       0   484.5      .1       0
Bank Sta=468.5,484.5
XS Rating Curve= 0 ,0
Exp/Cntr=0.3,0.1

Type RM Length L Ch R = 1 ,16698.6 ,182.2,164.9,146.5
XS GIS Cut Line= 4
     1766823.962       87058.139     1766945.574       86690.446
     1767108.064       86543.431     1767167.446       86201.884
#Sta/Elev= 30
     9.9 2128.48    49.7 2120.16    89.4 2123.73   119.2 2112.23   158.9 2110.41
   168.8 2098.45   188.7  2092.6   208.5 2074.03   228.4 2066.86   248.3 2047.67
   268.1 2042.38     278    2028   297.9 2021.14   317.8 2000.81   337.6 1998.02
   357.5 1983.72   454.5 1962.96     467 1962.19   479.5  1962.6   586.5 1977.48
   616.3 1976.56   626.2 1984.02     646 1985.98   665.8 1997.78   715.4 2005.73
   735.2 2017.13   774.8 2026.31   834.2 2030.62   883.7  2019.7   953.1 2024.68
#Mann= 3 , 0 , 0
       0      .1       0   454.5    .045       0   479.5      .1       0
Bank Sta=454.5,479.5
XS Rating Curve= 0 ,0
Exp/Cntr=0.3,0.1

Type RM Length L Ch R = 1 ,16533.7 ,296,293.8,287.8
XS GIS Cut Line= 4
     1767137.013       87087.857     1767115.802       86814.247
     1767150.621       86593.726     1767204.784       86206.845
#Sta/Elev= 30
     9.8 2034.95    29.4 2029.93      49 2028.38    58.8  2023.4    78.4 2021.04
   166.6 1997.04     245 1988.15   264.6  1982.3   284.1  1980.9   303.6  1967.3
     323 1965.58   332.7  1961.4   368.7 1958.98   381.2 1958.78   393.7 1959.74
     420 1961.53   439.4 1966.97   458.9 1967.73   468.6 1971.25   537.8 1979.52
     658 1987.73     678 1996.78     708 1999.39   758.1 1998.95   798.2 2005.55
   828.2  2012.8   848.3  2026.1   868.3  2032.9   878.3  2040.3   888.3 2043.31
#Mann= 3 , 0 , 0
       0      .1       0   368.7    .045       0   393.7      .1       0
Bank Sta=368.7,393.7
XS Rating Curve= 0 ,0
Exp/Cntr=0.3,0.1

Type RM Length L Ch R = 1 ,16240   ,221.4,225.8,230.2
XS GIS Cut Line= 5
     1767405.017       87191.777     1767444.995        86939.82
     1767377.892       86739.594      1767350.59       86463.322
     1767307.049       86217.297
#Sta/Elev= 30
     9.8 2127.12    88.3 2120.56     157 2105.58     206 2088.28   225.7 2087.15
   235.5 2078.25   255.1 2076.55   275.2 2062.76   325.5 2043.41   345.6  2024.1
   365.7 2022.56   375.8 2011.26   395.9 2006.32     416 1990.58   436.1 1987.07
   456.2 1973.04     543 1952.83   555.5 1951.61     568 1952.24   644.7 1974.73
   654.7 1983.99   674.5 1984.25   684.4 1997.84   704.2 2002.58   724.1 2020.38
   743.9 2024.12   753.9 2040.24   873.8 2063.95   933.8 2081.01   993.7 2083.49
#Mann= 3 , 0 , 0
       0      .1       0     543    .045       0     568      .1       0
Bank Sta=543,568
XS Rating Curve= 0 ,0
Exp/Cntr=0.3,0.1

Type RM Length L Ch R = 1 ,16014.2 ,86.4,88.5,90.5
XS GIS Cut Line= 4
     1767492.528       87131.612     1767583.927       86763.953
      1767607.14       86500.874     1767630.353       86268.746
#Sta/Elev= 30
      10 2101.22   159.5 2064.94   179.5 2050.68   239.3 2028.36   249.2 2018.64
   269.2  2012.8   289.1 1995.89     319 1983.83   378.8 1972.48   427.8 1952.84
   454.4 1949.69   466.9 1948.64   479.4 1950.29     506 1957.68   564.7 1985.85
   574.5 1985.86     594 2000.84   613.6 2004.87   633.2  2020.1     643 2020.87
   662.4 2038.73   681.8 2038.61   691.6 2054.29     711 2057.71   730.4 2073.81
     779 2091.65   798.5 2109.25   847.1 2131.01   866.5 2149.18   876.2 2149.17
#Mann= 3 , 0 , 0
       0      .1       0   454.4    .045       0   479.4      .1       0
Bank Sta=454.4,479.4
XS Rating Curve= 0 ,0
Exp/Cntr=0.3,0.1

Type RM Length L Ch R = 1 ,15925.7 ,285.2,283.3,281.4
XS GIS Cut Line= 4
     1767590.029       87154.294     1767657.434       86798.772
     1767715.466       86493.137     1767730.942       86295.828
#Sta/Elev= 30
    10.1 2102.07     191 2053.99     201 2041.11   221.1 2038.76   241.2 2020.03
   261.3 2015.65   271.4 2002.37   291.5 2001.01   311.6 1984.68     392 1963.79
   422.1 1947.51   432.1 1946.03   444.6 1946.22   492.3 1946.83   512.4 1961.16
   562.6 1975.28   582.6 1987.34   602.7 1988.47   612.7 1999.55   632.8 2002.22
   652.9 2016.26     673  2019.7   682.8 2031.14   702.6 2032.29   712.5  2042.9
   771.9 2067.54   781.8 2078.33   801.6 2083.61   821.4 2100.41   870.9 2123.96
#Mann= 3 , 0 , 0
    10.1      .1       0   422.1    .045       0   444.6      .1       0
#XS Ineff= 2 , 0
                          447.67         1964.05
Permanent Ineff=
       F       F
Bank Sta=422.1,444.6
XS Rating Curve= 0 ,0
Exp/Cntr=0.3,0.1

Type RM Length L Ch R = 1 ,15642.4 ,278.2,275.5,272.7
XS GIS Cut Line= 4
     1767820.696       87208.185     1767932.119       86891.623
      1767963.07       86562.775     1767986.282       86334.516
#Sta/Elev= 30
     9.9 2095.21    39.5 2087.04    98.7 2086.29   128.3 2065.73   148.1 2064.66
   236.9 2007.75   256.6 2004.71   276.4 1985.14   325.7 1969.04   345.6 1952.44
   433.2  1938.8   445.7 1938.08   458.2 1938.39   535.8 1951.31   545.8 1960.81
   565.8 1963.33   575.8 1973.44   595.8 1979.58   615.9 1994.74   635.9 1996.75
   645.9 2008.18   665.9  2009.7   715.8 2034.14   735.7 2035.11   745.7 2045.31
   765.7 2047.49   815.5 2070.93   835.5 2073.58   855.4 2085.35   895.3 2096.67
#Mann= 3 , 0 , 0
       0      .1       0   433.2    .045       0   458.2      .1       0
Bank Sta=433.2,458.2
XS Rating Curve= 0 ,0
Exp/Cntr=0.3,0.1

Type RM Length L Ch R = 1 ,15366.9 ,175.1,170.2,165.4
XS GIS Cut Line= 4
     1768110.578       87273.819     1768218.222       86994.929
     1768209.028       86562.788     1768235.677       86341.479
#Sta/Elev= 30
      10 2077.36    79.7 2073.29    89.7 2065.94   149.5 2062.16   199.3 2044.24
   219.2 2044.87   359.3 1987.19   379.4 1969.27   399.5 1965.85   409.5 1954.02
  477.27 1933.31   479.9 1931.34   492.4 1931.45   630.7 1941.03   650.8 1953.15
   670.9 1956.63   680.9 1967.83     701 1968.44   711.1 1980.02   731.2  1983.5
   750.6 1998.98   769.9 2001.72   779.6 2011.43     799 2013.96   818.4 2026.54
   866.9 2041.79   886.2 2055.76   905.6 2056.96   934.7  2068.8   954.1 2081.62
#Mann= 3 , 0 , 0
      10      .1       0  477.27    .045       0   492.4      .1       0
Bank Sta=477.27,492.4
XS Rating Curve= 0 ,0
Exp/Cntr=0.3,0.1

Type RM Length L Ch R = 1 ,15196.7 ,110.4,109.2,108
XS GIS Cut Line= 3
      1768415.72       87232.078     1768357.688       86682.708
     1768407.982       86380.941
#Sta/Elev= 30
      10  2140.6      30    2139    49.9  2122.4    69.9 2115.79    79.9 2104.31
    99.8 2100.34   109.8 2084.43   129.8 2076.97   149.8 2053.21   169.7 2044.98
   189.7 2027.28   199.7 2026.79   219.6 2010.33   299.5 1981.09   319.4 1966.66
   368.7 1952.82   388.5 1941.12   408.2 1939.55   425.3 1929.28   437.8 1928.83
   450.3 1929.25   506.9 1932.81     576  1947.3   615.5 1960.02   625.4 1971.66
   694.5 1996.35   822.7  2025.2   832.6 2033.23   852.4 2033.97   862.2 2040.52
#Mann= 3 , 0 , 0
      10      .1       0   425.3    .045       0   450.3      .1       0
#XS Ineff= 2 , 0
          424.84 1959.41
Permanent Ineff=
       F       F
Bank Sta=425.3,450.3
XS Rating Curve= 0 ,0
Exp/Cntr=0.3,0.1

Type RM Length L Ch R = 1 ,15087.5 ,164.3,185.3,206.3
XS GIS Cut Line= 4
     1768493.096        87224.34     1768516.309       86856.804
      1768446.67       86624.676      1768543.39       86361.597
#Sta/Elev= 30
      10 2132.12    59.7 2113.01    79.6 2096.47    89.6 2096.46   109.5 2069.44
   129.4 2061.23   139.3 2047.35   159.3 2038.63   179.2  2022.4   199.1  2018.5
   228.9 2003.69   278.7 1971.94   298.6 1970.66   308.5 1958.68   328.5  1956.8
   348.4 1944.41   378.4 1937.47   476.9 1927.38   489.4 1927.03   501.9  1928.9
   519.7 1938.86   580.3 1956.52   590.4 1964.68   610.6 1964.23   620.6 1973.85
   720.7 1995.16   770.8 2013.57   820.8 2021.95   850.9 2040.66   890.9 2056.68
#Mann= 3 , 0 , 0
       0      .1       0   476.9    .045       0   501.9      .1       0
Bank Sta=476.9,501.9
XS Rating Curve= 0 ,0
Exp/Cntr=0.3,0.1

Type RM Length L Ch R = 1 ,14902.1 ,71.5,71.3,71.2
XS GIS Cut Line= 4
     1768533.167       87234.402     1768574.341       86883.886
     1768740.699       86647.889     1768789.249       86324.449
#Sta/Elev= 30
    10.1 2127.12    70.6 2113.83    90.8 2094.43   100.8 2094.43     121 2064.66
   141.2 2055.35   191.6  2014.1   292.4 1961.38   362.9 1935.98   469.9 1919.21
   482.4 1918.59   494.9 1919.06   522.2 1934.19   542.1 1935.15   591.9    1955
   611.8 1973.24   631.7  1975.5   651.6 1992.37   730.9 2030.27   750.7 2046.89
   770.5 2049.72   800.2 2066.36   820.1 2085.48   839.9 2089.46   849.8 2112.44
   869.6 2115.27   889.4 2141.02   899.4 2142.29   919.2 2159.83   968.7 2178.14
#Mann= 3 , 0 , 0
       0     .08       0   469.9    .045       0   494.9      .1       0
Bank Sta=469.9,494.9
XS Rating Curve= 0 ,0
Exp/Cntr=0.3,0.1

Type RM Length L Ch R = 1 ,14830.8 ,183.3,162.6,141.9
XS GIS Cut Line= 4
     1768585.349       87196.152     1768660.959       86885.312
     1768770.173       86728.491     1768812.179       86409.249
#Sta/Elev= 30
      10 2095.85      50 2071.12      70 2068.76      80 2052.39     100  2046.6
     120 2023.98     140 2017.98     150 2002.27   169.9 1998.63   259.9  1948.8
     330 1924.43   397.9 1915.96   410.4 1915.41   422.9 1916.99   480.8 1934.29
   490.9 1944.96     511 1944.74   531.1 1961.16   581.4 1981.82   601.6 1997.79
   611.6 1997.82   682.1 2032.55   702.2 2049.28   722.3 2054.18   772.6 2090.72
   782.7 2091.48   792.8 2100.43   802.8 2120.29   822.9 2124.89     833 2141.65
#Mann= 3 , 0 , 0
       0     .08       0   397.9    .045       0   422.9      .1       0
Bank Sta=397.9,422.9
XS Rating Curve= 0 ,0
Exp/Cntr=0.3,0.1

Type RM Length L Ch R = 1 ,14668.2 ,227,227.5,228
XS GIS Cut Line= 4
      1768996.04       87216.603     1768891.582       86949.655
     1768821.944       86721.396     1768876.107        86384.81
#Sta/Elev= 30
     9.9 2040.93    39.5  2021.3    59.3 2020.87   128.5 1991.62   148.3 1975.72
     168 1975.98   177.9 1966.22     257 1936.48  359.59 1909.14   366.2 1907.49
   378.7 1907.57   485.5 1920.95   535.3  1949.5   555.4 1953.52   575.4  1970.3
   595.5 1974.08   605.5 1989.31   625.6 1991.87   635.6 2005.65   655.7 2012.79
   675.7 2030.47   695.8 2030.44   705.8 2047.27   725.8 2048.54   745.9 2067.95
   765.9 2075.55     776    2089     796 2092.73   806.1 2111.05   866.2 2145.78
#Mann= 3 , 0 , 0
     9.9      .1       0  359.59    .045       0   378.7      .1       0
Bank Sta=359.59,378.7
XS Rating Curve= 0 ,0
Exp/Cntr=0.3,0.1

Type RM Length L Ch R = 1 ,14440.7 ,52,58.8,65.6
XS GIS Cut Line= 5
      1769106.02       87317.574     1769138.731        87033.19
     1769058.797       86733.655     1769002.758       86546.183
     1768870.834       86294.784
#Sta/Elev= 30
     9.9 2132.91    59.2 2111.44    69.1 2098.38    88.8 2093.54   108.6 2074.17
   128.3 2070.67   138.2 2053.65   157.9 2054.05   167.8 2039.73   346.3  1950.6
   553.8 1901.81   566.3 1901.29   578.8 1903.94     743 1972.24   762.6 1994.29
   782.2 1998.35   801.7 2021.22   860.5 2056.86   880.1 2079.38   899.6 2084.31
   909.4 2104.35     929 2108.37   958.4  2136.4     978 2143.51   987.7 2157.21
  1007.3 2161.24  1026.9 2184.31  1046.5  2185.8  1066.1 2205.77  1075.9 2207.09
#Mann= 3 , 0 , 0
     9.9      .1       0   553.8    .045       0   578.8      .1       0
#XS Ineff= 2 , 0
          535.14 1936.63
Permanent Ineff=
       F       F
Bank Sta=553.8,578.8
XS Rating Curve= 0 ,0
Exp/Cntr=0.3,0.1

Type RM Length L Ch R = 1 ,14381.9 ,63.9,68,72.1
XS GIS Cut Line= 4
     1769209.831       87212.954     1769120.219       86851.707
      1769125.82       86633.279     1769013.805       86370.044
#Sta/Elev= 30
    10.1 2088.17    20.1 2085.42    70.4 2045.38   120.7 2022.91   140.8 2005.38
   191.1 1986.53   211.2 1970.71   231.4 1967.25   241.4 1954.88   382.1  1915.3
   449.1 1903.81   461.6 1901.27   474.1 1904.43   600.6 1940.59   620.3 1956.35
     640 1961.07   659.7 1978.54   679.5 1984.02   689.3 2001.48   709.1 2005.82
   728.8 2023.98   748.5  2032.3   768.3 2056.12     788 2056.29   797.9 2075.89
   817.6 2086.08   837.3 2108.43     857 2117.23   866.9 2126.41   876.8 2145.83
#Mann= 3 , 0 , 0
    10.1      .1       0   449.1    .045       0   474.1      .1       0
Bank Sta=449.1,474.1
XS Rating Curve= 0 ,0
Exp/Cntr=0.3,0.1

Type RM Length L Ch R = 1 ,14313.9 ,159.3,162.9,166.4
XS GIS Cut Line= 4
     1769262.988       87232.078     1769166.267       86880.017
     1769232.037       86566.644     1769208.824       86349.991
#Sta/Elev= 30
     9.9 2111.86    19.7 2100.07    39.5 2093.73    59.2 2068.68    69.1 2068.64
    88.8 2048.68   108.5 2041.98   128.3 2024.02     148 2022.25   157.9 2007.28
   177.6 2006.01   197.4 1990.35   335.5 1931.22   355.2  1930.2   435.1 1901.72
   472.7 1898.64   485.2 1898.51   495.2 1899.87   545.2 1916.78   595.2 1919.79
   665.3  1940.1   675.3 1949.32   764.5 1986.66   784.3 2003.26   804.2 2008.27
   833.9 2026.06   853.7  2045.1   873.5 2050.58   883.4 2067.13   903.2  2068.4
#Mann= 3 , 0 , 0
     9.9      .1       0   472.7    .045       0   495.2      .1       0
Bank Sta=472.7,495.2
XS Rating Curve= 0 ,0
Exp/Cntr=0.3,0.1

Type RM Length L Ch R = 1 ,14151.1 ,149.6,145.2,140.8
XS GIS Cut Line= 4
     1769305.544       87204.996     1769313.282       86895.492
     1769386.789       86702.052     1769359.708       86396.417
#Sta/Elev= 30
      10 2108.15      30  2081.3    39.9 2080.78    59.9    2055    79.9 2044.95
    99.9 2021.57   109.9 2021.17   129.8 2002.95   179.8 1982.67   199.7 1966.24
   219.7 1961.04   229.7 1948.79   249.7 1945.47   299.6 1913.74   319.5 1911.35
   329.3 1898.95   375.9 1887.78   388.4 1886.32   400.9  1887.2   427.8 1889.59
   437.7  1902.4   477.1 1916.13   536.3 1921.71   615.5 1945.73   635.3 1945.88
   645.2 1956.25     665 1958.07   684.8 1970.17     764 1993.15   823.4 2026.91
#Mann= 3 , 0 , 0
      10      .1       0   375.9    .045       0   400.9      .1       0
#XS Ineff= 2 , 0
                          412.04         1905.46
Permanent Ineff=
       F       F
Bank Sta=375.9,400.9
XS Rating Curve= 0 ,0
Exp/Cntr=0.3,0.1

Type RM Length L Ch R = 1 ,14005.9 ,202.9,195.9,188.9
XS GIS Cut Line= 4
      1769448.69        87290.11     1769460.412       86996.394
     1769506.722       86721.396     1769468.034        86384.81
#Sta/Elev= 30
     9.8 2085.59    29.4 2082.46      49 2065.74    68.6 2059.82    78.4 2047.42
      98 2045.17   107.8 2033.03     147 2012.31   264.6 1963.16   284.2 1947.29
   303.9 1944.96   313.9 1929.38   333.8 1925.63   353.7 1906.23   373.6 1900.95
   383.6 1887.74   420.9 1879.81   433.4 1879.14   445.9 1880.35   473.2 1884.37
   493.1 1900.29   562.9 1919.38   612.7 1921.36   712.3    1942   722.3 1952.35
   742.2 1954.39     792 1981.19     812 1982.44   821.9 1993.83   911.6 2034.32
#Mann= 3 , 0 , 0
       0      .1       0   420.9    .045       0   445.9      .1       0
Bank Sta=420.9,445.9
XS Rating Curve= 0 ,0
Exp/Cntr=0.3,0.1

Type RM Length L Ch R = 1 ,13809.9 ,238.4,237.3,236.3
XS GIS Cut Line= 4
     1769754.325       87255.291     1769696.293       86949.655
     1769661.474        86709.79     1769630.524       86419.629
#Sta/Elev= 30
      10 2061.84    30.1 2054.05    50.2  2033.2    70.2 2027.13    80.3 2017.62
   120.4  1996.2   140.5 1991.58   150.5 1979.57   170.6 1976.54   180.6 1965.61
   200.7 1959.19   220.8 1942.22   240.8  1940.3   250.9 1926.96     271  1925.5
     291 1908.89   301.1 1908.02   321.2 1895.09   371.7 1885.63   389.5 1876.69
     402 1874.61   414.5 1874.87   472.7 1879.88   513.1 1892.18   563.5 1917.96
   613.8 1923.39   744.7 1963.41   764.8 1974.01   784.9 1975.75   845.3 1994.21
#Mann= 3 , 0 , 0
       0      .1       0   389.5    .045       0   414.5      .1       0
Bank Sta=389.5,414.5
XS Rating Curve= 0 ,0
Exp/Cntr=0.3,0.1

Type RM Length L Ch R = 1 ,13572.6 ,324.6,316.8,309.1
XS GIS Cut Line= 4
      1769931.91       87284.757     1769942.849        86951.12
     1769870.335        86573.98     1769773.295       86349.479
#Sta/Elev= 30
     9.8 2065.15    78.5 2033.94   127.6 2018.78   147.3 2006.38   166.9 2003.97
   176.7  1994.7   235.6 1976.54   245.5 1967.02   265.1 1966.07   274.9 1956.37
   364.1 1925.87   384.3 1910.13   434.9  1890.6   455.1 1873.97     483 1865.79
   495.5 1863.37     508 1864.83   707.8  1896.9   727.6 1912.86   747.2 1916.79
   766.8 1932.55   786.3 1937.51   796.1  1952.2   815.7 1954.43   874.4  1991.7
     894  1992.5   903.7 2006.92   923.3 2014.81   942.9 2034.81   962.4 2041.65
#Mann= 3 , 0 , 0
       0      .1       0     483    .045       0     508      .1       0
Bank Sta=483,508
XS Rating Curve= 0 ,0
Exp/Cntr=0.3,0.1

Type RM Length L Ch R = 1 ,13255.8 ,97.6,96.6,95.7
XS GIS Cut Line= 4
     1770369.465       87100.539     1770261.139       86775.559
     1770133.468       86558.906      1769998.06       86315.172
#Sta/Elev= 30
    10.1 2010.41    40.3 2001.31    90.7 1997.53   120.9 1984.57   231.7 1965.55
     262 1953.95   282.1 1935.66   302.3 1929.63   312.3 1921.87   342.6 1914.51
   352.6 1904.12   402.9 1885.95     413 1877.39     423 1861.47   430.6  1857.9
   443.1 1855.39   455.6 1856.75   613.9 1873.84   623.9 1882.56   643.8 1885.87
   663.7  1898.2   683.7 1903.21   703.6 1918.57   723.5 1921.39   743.4  1939.2
   763.3  1941.1   773.3 1952.16   793.2 1958.91   823.1 1978.72   872.9 1993.58
#Mann= 3 , 0 , 0
       0      .1       0   430.6    .045       0   455.6      .1       0
Bank Sta=430.6,455.6
XS Rating Curve= 0 ,0
Exp/Cntr=0.3,0.1

Type RM Length L Ch R = 1 ,13159.1 ,170.8,171.2,171.6
XS GIS Cut Line= 4
     1770472.796       87044.932     1770324.377       86697.687
     1770209.562       86518.464     1770139.552       86246.828
#Sta/Elev= 30
     9.9 2072.89    59.6 2056.94    89.4 2036.98   139.1 2017.65     159 2003.07
   208.7  1987.7   228.6 1972.06   248.4 1970.24   268.3 1955.84   288.2 1948.67
   308.1 1930.22   327.9 1926.87   337.9 1910.62   357.8 1907.28   377.6 1885.92
     397 1880.65   406.7  1873.9   416.3 1860.79  446.61 1857.09     455 1854.52
   467.5 1855.24   590.5  1865.4   680.6 1886.87   700.7 1886.97   770.8 1912.89
   790.8 1928.51   800.9 1928.52   830.9 1943.45     861  1967.3     871 1969.15
#Mann= 3 , 0 , 0
     9.9     .08       0  446.61    .045       0   467.5      .1       0
Bank Sta=446.61,467.5
XS Rating Curve= 0 ,0
Exp/Cntr=0.3,0.1

Type RM Length L Ch R = 1 ,12988   ,335.6,334.2,332.8
XS GIS Cut Line= 4
      1770539.02       87049.571     1770531.901       86722.421
     1770298.364        86344.01     1770203.107       86183.632
#Sta/Elev= 30
     9.9 2109.25    29.7 2106.01    49.6 2087.43   128.9 2067.67   148.7 2049.98
   168.6 2042.67   188.4 2016.88   198.3 2016.88   267.7 1985.56   287.6 1969.95
   307.4 1966.52   337.3 1952.41   357.5 1934.69   377.8  1930.6     398 1906.46
   418.2 1905.23   428.3 1892.41   478.8 1859.39   509.1 1849.21   519.2 1848.05
   531.7 1848.11   620.3 1853.97   771.9 1883.56   791.5    1894   811.2 1896.97
   830.8  1916.5   850.4 1920.58   870.1 1934.48     929 1952.11   958.4 1954.92
#Mann= 3 , 0 , 0
     9.9     .08       0   509.1    .045       0   531.7     .08       0
Bank Sta=509.1,531.7
XS Rating Curve= 0 ,0
Exp/Cntr=0.3,0.1

Type RM Length L Ch R = 1 ,12653.8 ,419.4,427.6,435.9
XS GIS Cut Line= 4
     1770834.371       86901.895     1770858.885        86589.74
     1770549.959       86152.578     1770358.528       86010.372
#Sta/Elev= 30
    10.1 1975.05    50.5 1974.09   121.2 1963.88   333.3 1927.94   353.5 1913.67
   373.7 1909.78   393.9 1897.63   414.1 1894.53   434.3 1881.41   454.5 1879.36
   494.9 1860.71   515.1  1846.3   545.4 1840.39   603.6 1838.21   616.1 1838.07
   628.6 1838.74     707 1846.68   777.7 1863.92     808 1877.74   828.2 1881.79
   848.4 1895.09   878.2 1901.32   898.1 1913.75     918 1916.39   957.7 1938.94
   987.5 1944.73  1007.4 1961.87  1037.2  1965.3  1057.1 1979.29  1086.9 1984.31
#Mann= 3 , 0 , 0
       0     .08       0   603.6    .045       0   628.6      .1       0
Bank Sta=603.6,628.6
XS Rating Curve= 0 ,0
Exp/Cntr=0.3,0.1

Type RM Length L Ch R = 1 ,12226.1 ,227.8,236.6,245.3
XS GIS Cut Line= 4
     1771173.478       86737.811      1771149.87       86467.956
     1771042.211       86043.189     1770942.048       85785.146
#Sta/Elev= 30
      10 2122.82    30.1 2118.27    40.1 2104.61    60.2 2096.11    80.3 2075.52
   130.4 2049.79   150.5  2031.9   270.9 1975.75   320.7 1939.37   340.6 1934.85
   350.6 1918.01   370.5 1917.36     490 1834.08   517.3 1827.79   529.8 1825.61
   542.3 1826.23   649.3 1843.27     719 1872.25   738.7 1889.86   758.5 1893.53
   768.4 1909.15   788.2 1911.66   847.5 1956.42   867.3 1960.07   877.1 1976.13
   896.9 1980.21   916.7 2002.49   936.5 2008.81     976 2036.77   985.9 2057.71
#Mann= 3 , 0 , 0
       0      .1       0   517.3    .045       0   542.3      .1       0
Bank Sta=517.3,542.3
XS Rating Curve= 0 ,0
Exp/Cntr=0.3,0.1

Type RM Length L Ch R = 1 ,11989.6 ,135.1,125.6,116
XS GIS Cut Line= 4
     1771390.829        86613.07     1771297.978       86272.615
      1771325.06       86048.224     1771178.045        85769.67
#Sta/Elev= 30
    10.1 2063.97    20.2 2051.31    40.3 2048.97    60.5 2032.83   110.9 2016.93
   252.1 1951.53   272.2 1928.29   292.4 1923.12   302.5 1907.59   322.6 1905.98
   332.7 1890.19   352.9  1882.4   372.5 1861.87   441.3 1821.69   451.2 1820.35
   463.7 1821.64   559.3 1834.64     638 1857.96   647.8 1870.29   667.5 1873.28
   716.7 1897.43   726.5 1908.05   746.2 1912.71   765.9  1936.6   785.6  1939.4
   805.3 1966.47   844.7 2001.22   864.3 2003.37   874.2  2017.6   893.9 2025.59
#Mann= 3 , 0 , 0
    10.1     .08       0   441.3    .045       0   463.7      .1       0
Bank Sta=441.3,463.7
XS Rating Curve= 0 ,0
Exp/Cntr=0.3,0.1

Type RM Length L Ch R = 1 ,11864   ,211.8,201.9,192
XS GIS Cut Line= 4
     1771641.978       86565.239     1771503.024       86377.073
      1771386.96       86005.667     1771326.519       85691.035
#Sta/Elev= 30
     9.7 2017.61      39 2005.51    97.5 1968.27     117 1962.91   136.4 1947.29
   165.7 1939.98   175.4 1928.68   204.7 1925.53   263.8 1898.28   283.8 1896.46
   293.8 1883.58   313.7 1883.59   323.7 1873.32   440.9 1819.19   453.4  1818.4
   465.9 1818.93   593.1 1836.83   663.1 1855.06   683.1 1868.97   703.1 1873.61
   713.1 1884.84   733.2 1886.65   743.2  1900.2   763.2 1909.01   783.2 1931.22
   803.2 1939.38   823.3 1961.51   833.3  1962.2   853.3 1979.78   943.4 1971.83
#Mann= 3 , 0 , 0
       0     .08       0   440.9    .045       0   465.9     .08       0
Bank Sta=440.9,465.9
XS Rating Curve= 0 ,0
Exp/Cntr=0.3,0.1

Type RM Length L Ch R = 1 ,11662.1 ,182,181.7,181.3
XS GIS Cut Line= 4
     1771862.823       86411.892     1771653.908       86113.994
     1771495.287       85939.898      1771386.96       85665.213
#Sta/Elev= 30
    10.1 2000.29    20.2 1996.15    40.4 1978.74    60.6 1973.69   161.7 1910.88
   181.9 1904.11   202.1  1888.1   222.4 1886.78   232.5    1873   242.6 1867.65
   262.8 1864.24     283 1850.57   303.2 1847.54   323.4 1837.16   343.6 1836.13
   363.9 1825.89   439.7 1810.96   452.2 1810.13   464.7 1811.05   560.1 1823.96
   609.2 1839.24   628.9  1858.9   648.6  1861.9   658.4 1877.95   678.1  1884.1
   707.6 1912.73   796.2 1933.56   815.9 1929.96   865.1 1934.59   894.6 1928.49
#Mann= 3 , 0 , 0
       0     .08       0   439.7    .045       0   464.7      .1       0
Bank Sta=439.7,464.7
XS Rating Curve= 0 ,0
Exp/Cntr=0.3,0.1

Type RM Length L Ch R = 1 ,11480.4 ,142,141.8,141.5
XS GIS Cut Line= 4
     1771939.203       86376.826     1771858.399       86079.753
     1771627.444       85818.941     1771430.543       85594.693
#Sta/Elev= 30
     9.9 2013.39    29.8 1999.18    49.7 1994.72    59.6 1983.24    79.4 1977.13
    99.3 1961.39     149 1944.61   168.8  1926.9   198.6 1909.89   228.4 1899.96
   238.3  1890.1   258.2 1888.37   268.1 1876.65     288 1869.48   307.9 1852.92
   327.8 1848.39   347.7 1832.19   377.5 1824.58   397.4 1810.63   454.6 1808.94
   467.1 1807.72   479.6 1808.65   556.7 1810.99   656.2 1827.27   775.6  1852.7
   845.2 1873.51     895  1875.7   914.9 1886.06   934.8 1882.16   954.7 1889.37
#Mann= 3 , 0 , 0
     9.9     .08       0   454.6    .045       0   479.6      .1       0
#XS Ineff= 2 , 0
          428.93 1835.49   504.6         1834.44
Permanent Ineff=
       F       F
Bank Sta=454.6,479.6
XS Rating Curve= 0 ,0
Exp/Cntr=0.3,0.1

Type RM Length L Ch R = 1 ,11338.7 ,174.6,176.4,178.2
XS GIS Cut Line= 4
     1772157.982       86294.784     1772032.184       86048.658
     1771709.486       85715.021     1771557.188       85514.329
#Sta/Elev= 30
     9.9 1978.58    19.7 1971.63    39.5 1972.96    49.4 1962.41    69.1 1960.46
    88.8 1948.13   108.6 1944.68   118.5 1940.04   128.3 1929.03   148.1 1926.58
   167.8 1913.03   187.6 1912.67   207.3 1901.38   227.1 1899.21   246.8 1889.89
   266.5 1888.31   276.4 1872.14   306.7 1869.62   326.9 1856.43     347 1854.15
   377.3 1841.03   397.5  1839.4   518.6 1801.11   528.7 1798.62   541.2 1798.72
   629.6 1801.71   760.7 1816.86   811.1 1819.81   871.6 1816.37   992.5 1827.72
#Mann= 3 , 0 , 0
     9.9     .08       0   518.6    .045       0   541.2     .08       0
#XS Ineff= 2 , 0
                          588.47         1820.05
Permanent Ineff=
       F       F
Bank Sta=518.6,541.2
XS Rating Curve= 0 ,0
Exp/Cntr=0.3,0.1

Type RM Length L Ch R = 1 ,11162.3 ,98.7,97.3,95.9
XS GIS Cut Line= 4
      1772261.31       86086.912     1772119.883       85915.314
     1771843.302        85579.73     1771627.444       85397.792
#Sta/Elev= 30
    10.1 1970.74    40.4 1957.91    60.6 1957.74    80.9 1945.24   101.1 1945.26
   121.3 1933.27   141.5 1932.72   171.8 1918.39     192 1917.79   232.5 1905.91
   303.3 1859.68   313.4  1847.7   374.1 1814.91   404.4 1805.65   462.7 1796.92
   475.2 1796.64   487.7  1796.7   606.7 1805.46   667.3 1820.95   697.6 1823.81
   717.7 1834.37     748 1832.79   768.1 1847.48   798.4 1848.23   828.6 1856.39
   848.8 1852.38     869  1859.4   889.1 1854.06   919.4 1858.68   939.5 1857.17
#Mann= 3 , 0 , 0
       0     .08       0   462.7    .045       0   487.7     .08       0
Bank Sta=462.7,487.7
XS Rating Curve= 0 ,0
Exp/Cntr=0.3,0.1

Type RM Length L Ch R = 1 ,11065   ,197.6,201,204.3
XS GIS Cut Line= 4
     1772387.699       86141.639     1772141.573       85775.185
     1771855.086       85467.904     1771739.021       85328.627
#Sta/Elev= 30
      10  2035.2    20.1  2026.5   150.5 2002.85   170.6 1992.06   200.7    1991
   220.7 1978.39   250.8 1974.26     301 1948.81     321 1924.62   341.1 1923.11
   361.2 1898.62   381.2 1893.45   411.3 1866.55   501.5 1817.91   581.5 1795.66
     609 1794.51   621.5 1794.43     634 1794.45   691.5 1799.01   741.5 1810.82
   761.5 1823.22   791.5 1827.47   801.5 1836.85   831.5 1845.15   861.6 1866.84
   881.7 1870.47   901.8 1891.45     922 1891.57   942.1 1905.52  1042.9 1920.19
#Mann= 3 , 0 , 0
       0      .1       0     609    .045       0     634      .1       0
Bank Sta=609,634
XS Rating Curve= 0 ,0
Exp/Cntr=0.3,0.1

Type RM Length L Ch R = 1 ,10864.1 ,201.7,216.7,231.7
XS GIS Cut Line= 4
     1772431.455       85983.025     1772318.519       85730.116
     1772032.184        85315.75     1771851.692       85184.483
#Sta/Elev= 30
     9.9  2059.2    29.7 2057.38    59.4 2040.25      89 2015.56   108.8 2009.31
   118.7 1992.87   138.5 1987.88   158.3 1968.91   217.6 1935.36   227.5 1921.77
   247.3 1918.84   267.1 1899.64   347.5 1852.04   407.9 1830.23   428.1 1815.46
   536.5 1787.74     549 1786.19   561.5 1787.05   649.7 1805.39     690 1825.09
   710.1 1850.07   740.4 1859.28   750.4 1876.04   780.7 1889.35   800.1  1910.8
   819.5 1916.19   916.5 1977.28   945.6 1983.63     965 2003.08  1003.8 2012.29
#Mann= 3 , 0 , 0
       0      .1       0   536.5    .045       0   561.5      .1       0
Bank Sta=536.5,561.5
XS Rating Curve= 0 ,0
Exp/Cntr=0.3,0.1

Type RM Length L Ch R = 1 ,10647.3 ,221.2,219.5,217.8
XS GIS Cut Line= 4
      1772520.52       85874.128     1772354.161       85529.805
     1772369.636       85258.988     1772191.671       85046.204
#Sta/Elev= 30
    10.1 2037.27    40.3 2015.46    60.4 2010.55    80.5 1995.87   100.6 1988.89
   110.7 1978.13   130.8 1975.91   150.9 1954.89   191.2 1924.35   211.3 1914.67
   221.4 1897.12   241.5  1893.6   301.9  1849.7     322 1845.51   332.1 1832.75
   362.3 1819.07   372.3 1807.38   412.5 1791.14   470.4 1781.75   482.9  1779.9
   495.4 1779.96   563.2 1784.63   573.3 1793.06   593.4  1795.4   613.5 1806.65
   713.1 1831.26   782.5 1860.29   841.9  1878.1   871.6 1901.89   931.1 1915.03
#Mann= 3 , 0 , 0
       0     .08       0   470.4    .045       0   495.4     .08       0
Bank Sta=470.4,495.4
XS Rating Curve= 0 ,0
Exp/Cntr=0.3,0.1

Type RM Length L Ch R = 1 ,10427.8 ,246.4,256.2,266.1
XS GIS Cut Line= 4
     1772575.588       85871.732     1772579.591       85514.255
     1772574.683       85251.251     1772448.338       84956.274
#Sta/Elev= 30
     9.9    2029    69.5 1984.97    89.4 1981.23    99.3 1966.93   119.2 1964.22
     139 1947.16     149 1946.59   168.8  1924.6   188.7 1923.91   198.6 1902.11
   218.5 1899.92   238.3 1877.84   258.2  1871.8   268.1 1860.37     288 1858.21
   297.9 1846.56   386.7 1810.04   406.2 1792.98   461.9 1775.93   474.4 1773.41
   486.9 1773.62   552.4 1782.23   591.3 1795.46   610.8 1809.46     791 1852.16
   811.1 1850.28   821.1 1859.09   881.3 1873.17   901.3 1885.14   941.4 1891.53
#Mann= 3 , 0 , 0
       0      .1       0   461.9    .045       0   486.9      .1       0
Bank Sta=461.9,486.9
XS Rating Curve= 0 ,0
Exp/Cntr=0.3,0.1

Type RM Length L Ch R = 1 ,10171.6 ,199,196.1,193.2
XS GIS Cut Line= 4
     1772675.272       85885.735     1772775.861       85529.805
     1772880.318       85289.939     1772864.843       85050.073
#Sta/Elev= 30
      10 2043.06      30 2038.46      50 2017.57      70  2012.1      90 1993.98
     100 1995.25     120 1975.96     140 1969.69   159.9 1946.34   179.9 1937.31
   189.9  1918.4   209.9 1917.66   219.9 1897.97   279.9 1863.53   299.9 1841.99
   309.9 1840.77   329.9 1822.54   349.9 1817.15   369.9 1798.87     390  1794.1
   400.1 1780.74   447.9 1769.14   460.4 1768.55   472.9 1768.78   530.9 1774.02
   571.1 1789.24   591.2  1804.4   711.6 1831.58   811.8 1872.88   871.9 1905.16
#Mann= 3 , 0 , 0
       0     .08       0   447.9    .045       0   472.9     .08       0
Bank Sta=447.9,472.9
XS Rating Curve= 0 ,0
Exp/Cntr=0.3,0.1

Type RM Length L Ch R = 1 ,9975.5  ,262,265.2,268.4
XS GIS Cut Line= 4
     1772759.623       85993.964     1772945.585       85687.674
     1773058.428       85298.709     1773128.272       85076.186
#Sta/Elev= 30
      10 2080.12    39.8 2068.12    59.7 2050.69    79.6 2045.98   109.5 2020.07
   129.4  2014.8   149.3  1987.5     209 1946.34     219 1929.67   238.9 1923.01
   268.7 1894.77   288.6 1889.21   308.6 1868.26   328.5 1864.86   338.4 1851.42
   378.1 1830.35   437.3 1809.15   447.2 1796.35     467  1794.6   486.7  1780.5
   526.3 1767.42   553.3    1766   565.8  1765.8   578.3  1768.6   664.5  1803.8
   753.4 1829.52   763.3 1841.72   782.8 1842.99   889.7 1880.93   996.6    1934
#Mann= 3 , 0 , 0
       0     .08       0   553.3    .045       0   578.3     .08       0
Bank Sta=553.3,578.3
XS Rating Curve= 0 ,0
Exp/Cntr=0.3,0.1

Type RM Length L Ch R = 1 ,9710.3  ,291,289.3,287.7
XS GIS Cut Line= 4
     1772934.646       86037.719     1773152.595       85807.626
       1773301.1       85479.834     1773426.898       85146.197
#Sta/Elev= 30
     9.9 2043.66    29.7 2038.11    49.5 2018.82    69.3 2016.56      99 1983.48
   118.8 1976.84   138.7 1944.14   168.4 1936.75   188.2 1907.35     208 1903.48
   237.7 1877.46   267.4 1865.77   287.2 1848.52   396.9 1793.14   476.9 1764.62
   514.4 1762.96   526.9 1762.88   539.4  1763.3   566.8 1764.42   656.8 1805.87
   716.4  1816.7   855.1 1868.62   914.5 1905.33   934.3  1908.6   944.2 1925.64
     964 1930.77   983.8 1952.34  1003.6  1959.5  1023.5 1984.42  1033.4 1985.45
#Mann= 3 , 0 , 0
       0     .08       0   514.4    .045       0   539.4     .08       0
Bank Sta=514.4,539.4
XS Rating Curve= 0 ,0
Exp/Cntr=0.3,0.1

Type RM Length L Ch R = 1 ,9421    ,367.6,362,356.3
XS GIS Cut Line= 4
     1773147.955       86163.517     1773431.528       85926.001
     1773561.461       85574.032     1773646.341       85344.102
#Sta/Elev= 30
      10 1960.11      40 1934.71      60 1922.44      70 1921.84     100 1899.09
     180 1870.05   199.9 1857.49   219.9  1855.5   279.9 1830.13   309.9 1812.47
   448.9 1784.48   458.8 1779.47   468.6 1765.44   574.6  1756.4   577.2 1755.83
   599.6 1757.09   666.1 1774.34   685.8 1796.74   705.6 1800.09   725.3 1816.97
   745.1 1823.36   764.7 1838.42   774.5 1838.78   813.7  1856.9   833.3 1873.11
   862.7 1886.38   882.3 1889.31   911.8 1915.33   960.8 1933.12   990.2  1949.4
#Mann= 3 , 0 , 0
       0     .08       0   574.6    .045       0   599.6     .08       0
Bank Sta=574.6,599.6
XS Rating Curve= 0 ,0
Exp/Cntr=0.3,0.1

Type RM Length L Ch R = 1 ,9059    ,295.4,293.3,291.3
XS GIS Cut Line= 4
     1773683.962       86327.601     1773798.821       86081.475
     1773842.675       85648.357     1773886.207       85421.478
#Sta/Elev= 30
    10.1 1930.31    30.2 1911.13    50.3 1904.08    60.4 1890.46    80.5 1885.28
   100.6 1865.17   120.7 1858.85   140.8 1841.09     161 1837.07   181.1 1817.58
   201.2 1813.47   251.5 1780.98   390.3 1752.27   447.1 1748.53   459.6 1747.91
   472.1 1748.53   489.3 1759.97   509.1 1759.98   677.3 1820.14     697 1833.43
   787.3 1867.84   797.3 1879.73   817.4 1881.81   827.5 1895.77   847.6 1902.47
   867.6 1927.37   887.7 1929.22   897.8 1951.27   917.9 1951.81     938 1975.34
#Mann= 3 , 0 , 0
       0     .08       0   447.1    .045       0   472.1     .08       0
Bank Sta=447.1,472.1
XS Rating Curve= 0 ,0
Exp/Cntr=0.3,0.1

Type RM Length L Ch R = 1 ,8765.7  ,335.2,325.7,316.2
XS GIS Cut Line= 3
     1774160.892       86315.172     1774098.991       86044.356
     1773959.714       85452.429
#Sta/Elev= 30
     9.9 1884.63   109.1 1850.93   119.1 1839.07   138.9 1835.86   148.8 1822.38
   158.7 1816.61   208.4 1797.91   228.2 1783.37   238.1 1782.62     258 1766.76
   277.8  1761.2   297.8 1749.39   355.5 1744.41     368 1744.03   380.5 1744.35
   448.2 1751.09   458.2 1757.08   478.3 1758.73   597.5 1806.59   726.4 1841.89
   746.2 1854.47   766.1 1854.57     776 1865.45   795.8  1870.3   815.7    1885
   835.5  1891.4   855.3 1913.35   875.2 1914.53   885.1 1938.95     895 1943.43
#Mann= 3 , 0 , 0
     9.9     .08       0   355.5    .045       0   380.5     .08       0
#XS Ineff= 2 , 0
          326.31 1764.47
Permanent Ineff=
       F       F
Bank Sta=355.5,380.5
XS Rating Curve= 0 ,0
Exp/Cntr=0.3,0.1

Type RM Length L Ch R = 1 ,8440    ,329.8,332.3,328.9
XS GIS Cut Line= 4
     1774473.372       86291.547     1774442.928       85995.609
     1774309.841       85689.199     1774114.051       85408.023
#Sta/Elev= 30
     9.9 2005.71    49.6 1980.05    59.5 1967.32    79.3 1962.31    99.2 1938.15
   109.1 1937.25   168.6 1886.87   178.5 1886.19   198.3 1863.79   218.2 1858.04
   267.8 1825.24   287.6 1822.93   297.5 1809.99   317.2 1808.53   376.1 1772.21
   395.8 1770.96   405.6 1757.53   454.7 1742.48     511 1738.89   523.5 1738.12
     536 1738.74   671.9 1796.73     813 1835.11   853.3 1854.13   873.4 1876.67
   893.6 1877.36   913.7 1896.72   933.9 1900.15     954 1918.22   974.2 1924.79
#Mann= 3 , 0 , 0
       0     .08       0     511    .045       0     536     .08       0
Bank Sta=511,536
XS Rating Curve= 0 ,0
Exp/Cntr=0.3,0.1

Type RM Length L Ch R = 1 ,8107.6  ,228,243.5,259
XS GIS Cut Line= 4
     1774590.329       86276.484     1774656.486       85899.662
     1774523.399       85723.245     1774489.741       85355.709
#Sta/Elev= 30
    10.1 1978.32    30.2 1969.24    50.3 1948.92    70.5 1945.08    80.5 1930.88
   100.7 1926.26   120.8 1904.71     141 1898.54     151 1884.46   171.2  1883.8
   181.2 1869.06   201.4  1865.3   221.5 1848.11   241.6 1843.73   251.7 1830.17
   271.8 1827.66     292 1809.65   392.6 1766.57   412.7 1763.91     473 1737.47
   490.6 1734.69   503.1 1734.17   515.6 1737.37   623.5 1741.32   723.3 1764.19
   793.1 1793.04   803.1 1808.07     843 1831.03   872.9 1840.94   972.6 1852.96
#Mann= 3 , 0 , 0
       0     .08       0   490.6    .045       0   515.6     .08       0
Bank Sta=490.6,515.6
XS Rating Curve= 0 ,0
Exp/Cntr=0.3,0.1

Type RM Length L Ch R = 1 ,7864.2  ,387.6,386.9,345
XS GIS Cut Line= 3
     1774710.262       86261.008     1774799.245       85874.128
     1774803.114       85347.971
#Sta/Elev= 30
     9.9 1950.64    19.8 1947.89    29.8 1933.37    49.6 1928.07    69.5 1907.17
    89.3 1899.29   109.2 1884.88   119.1 1884.08   138.9 1868.08   158.8 1865.05
   168.7 1853.75   188.6 1848.34   208.4 1832.57   228.3 1829.65   238.2 1818.26
     258 1815.73   317.6 1781.55   327.5  1780.4   347.4 1765.58   367.2 1763.07
   377.1 1753.94   416.9 1740.18   484.2 1733.05   496.7 1732.87   509.2 1733.89
   636.3 1743.45   685.9 1756.53     765  1768.5     854 1790.43   923.2 1794.33
#Mann= 3 , 0 , 0
       0     .08       0   484.2    .045       0   509.2     .08       0
Bank Sta=484.2,509.2
XS Rating Curve= 0 ,0
Exp/Cntr=0.3,0.1

Type RM Length L Ch R = 1 ,7477.2  ,206.4,213.2,220.1
XS GIS Cut Line= 4
     1774772.826       86291.116     1775035.242       85990.192
      1775073.93       85630.394      1775070.35       85370.676
#Sta/Elev= 30
      10 1947.63   139.7 1868.62   159.7 1863.92   179.7 1848.68   199.6 1845.84
   219.6 1830.67   239.6 1827.89   309.4 1794.51   449.5 1756.02   469.6 1742.56
   497.3 1735.13   509.8 1731.83   522.3 1732.51   620.4 1750.09   670.7 1775.89
   690.8 1780.36     741 1812.66   761.1  1816.5   771.1 1826.61   831.1 1847.25
   841.1 1856.99     861  1857.8     871 1868.11     891  1870.5     941 1894.71
   960.9 1894.68   970.9  1904.7   990.9 1907.31  1010.9  1921.9  1020.9 1922.57
#Mann= 3 , 0 , 0
       0     .08       0   497.3    .045       0   522.3     .08       0
Bank Sta=497.3,522.3
XS Rating Curve= 0 ,0
Exp/Cntr=0.3,0.1
